--- HurrcneCrk.prj (project) ---

Proj Title=HurrcneCrk
Current Plan=p01
Default Exp/Contr=0,0
English Units
Geom File=g01
Flow File=f01
Plan File=p01
BEGIN DESCRIPTION:
AMEC Environment & Infrastructure, 2013
Projection: NAD 1983 State Plane West Virginia South FIPS 4702 (US Feet)
Vertical Datum: NAVD 1988
END DESCRIPTION:
DSS File=dss
DSS Export Rating Curves= 0
DSS Export Rating Curve Sorted= 0
DSS Export Volume Flow Curves= 0
DXF OffsetX= 0
DXF OffsetY= 0
DXF ScaleX= 0
DXF ScaleY= 0

--- HurrcneCrk.p01 (plan) ---

Plan Title=Floodplain
Program Version=4.10
Short Identifier=Floodplain
Geom File=g01
Flow File=f01
Subcritical Flow
K Sum by GR= 0
Std Step Tol= 0.01
Critical Tol= 0.01
Num of Std Step Trials= 20
Max Error Tol= 0.3
Flow Tol Ratio= 0.001
Split Flow NTrial= 30
Split Flow Tol= 0.02
Split Flow Ratio= 0.02
Log Output Level= 0
Friction Slope Method= 1
Unsteady Friction Slope Method= 2
Unsteady Bridges Friction Slope Method= 1
Parabolic Critical Depth
Global Vel Dist= 0 , 0 , 0
Global Log Level= 0
CheckData=True
Encroach Param=-1 ,0,0, 0
Run HTab= 0
Run UNet= 0
Run PostProcess= 0
Run WQNet= 0
UNET Theta= 0
UNET Theta Warmup= 0
UNET ZTol= 0
UNET ZSATol= 0
UNET MxIter= 0
UNET MaxInSteps= 0
UNET DtIC= 0
UNET DtMin= 0
UNET MaxCRTS= 0
UNET WFStab= 0
UNET SFStab= 0
UNET WFX= 1
UNET SFX= 1
UNET DSS MLevel= 1
UNET DZMax Abort= 0
UNET Convert EG Bridges= 0
UNET Use Existing IB Tables= 0
UNET Froude Reduction=False
UNET Froude Limit= 0
UNET Froude Power= 0
UNET Time Slicing=0,0, 5
UNET Junction Losses=0
DSS File=dss
Write IC File= 0
Write IC File at Sim End=0
Echo Input=False
Echo Parameters=False
Echo Output=False
Write Detailed= 0
WQ AD Non Conservative
WQ ULTIMATE=-1
WQ Max Comp Step=1HOUR
WQ Output Interval=15MIN
WQ Output Selected Increments= 0
WQ Output face flow=0
WQ Output face velocity=0
WQ Output face area=0
WQ Output face dispersion=0
WQ Output cell volume=0
WQ Output cell surface area=0
WQ Output cell continuity=0
WQ Output cumulative cell continuity=0
WQ Output face conc=0
WQ Output face dconc_dx=0
WQ Output face courant=0
WQ Output face peclet=0
WQ Output face adv mass=0
WQ Output face disp mass=0
WQ Output cell mass=0
WQ Output cell source sink temp=0
WQ Output cell source sink nsm=0
WQ Output MaxMinRange=-1
WQ Daily Max Min Mean=-1
WQ Daily Range=0
WQ Daily Time=0
WQ Create Restart=0
WQ Fixed Restart=0
WQ System Summary=0
WQ Use Fixed Temperature=0
Sorting and Armoring Iterations= 10
XS Update Threshold= 0.02
Hydraulics Update Threshold= 0.02
Energy Slope Method= 1
Volume Change Method= 0
XS Weighting Method= 0
Number of US Weighted Cross Sections= 1
Number of DS Weighted Cross Sections= 1
Upstream XS Weight=0.25
Main XS Weight=0.5
Downstream XS Weight=0.25
Number of DS XS's Weighted with US Boundary= 1
Upstream Boundary Weight= 1
Weight of XSs Associated with US Boundary= 0
Number of US XS's Weighted with DS Boundary= 1
Downstream Boundary Weight= 0.5
Weight of XSs Associated with DS Boundary= 0.5
Sediment Output Level= 4
Mass or Volume Output= 0
Output Increment Type= 1
Profile and TS Output Increment= 10
XS Output Flag= 0
XS Output Increment= 10
Disregard all LS=0
Disregard all Conn=0
Disregard all Breaches=0
Disregard all Pumps=0

--- HurrcneCrk.f01 (steady flow) ---

Flow Title=NFF Regression Equation
Program Version=4.10
Number of Profiles= 1
Profile Names=P100yr
River Rch & RM=HurrcneCrk,Main            ,27000.5
1099.669
River Rch & RM=HurrcneCrk,Main            ,25495.9
1126.260
River Rch & RM=HurrcneCrk,Main            ,23781.1
1248.928
River Rch & RM=HurrcneCrk,Main            ,23443.6
1456.393
River Rch & RM=HurrcneCrk,Main            ,19734.3
1517.867
River Rch & RM=HurrcneCrk,Main            ,14454.6
1686.299
River Rch & RM=HurrcneCrk,Main            ,14117.8
1878.896
River Rch & RM=HurrcneCrk,Main            ,9667.1
2014.925
River Rch & RM=HurrcneCrk,Main            ,1336.7
2231.218
River Rch & RM=HurrcneCrk,Main            ,980.6
3661.633
River Rch & RM=HurrcneCrk,Main            ,672.9
4769.873
River Rch & RM=HurrcneCrk,Main            ,350.7
4770.603
River Rch & RM=HurrcneCrk,Main            ,8.8
5204.667
Boundary for River Rch & Prof#=HurrcneCrk,Main            , 1
Up Type= 0
Dn Type= 3
Dn Slope=0.00329
DSS Import GetInterval= 0
DSS Import GetPeak= 0
DSS Import FillOption= 0

--- HurrcneCrk.g01 (geometry) ---

Geom Title=USGS 3m DEM
Program Version=4.10

River Reach=HurrcneCrk      ,Main
Reach XY= 30
     1882230.524      575749.326     1882180.603      575410.667
     1881546.102       574798.41     1881151.259      572388.342
     1879777.775       571332.39     1879864.629      570679.393
     1880326.606      570161.869     1880449.924      569715.541
     1880038.348      568923.595     1880014.053      568275.805
     1879586.844      567595.008      1878864.38       567509.89
     1878713.486      567833.841     1877480.223      567817.246
     1877188.466       567548.05     1876999.237      566675.548
     1876080.496      566064.879     1875795.669      566382.687
     1874965.518      566726.528     1874635.723      567250.808
     1874328.134      567308.303     1873998.172      566959.217
     1873291.334      567049.504     1872879.748      566695.207
     1872452.523      566606.622     1872132.992      565943.196
     1872237.212      565286.728     1871790.907      564446.155
     1868856.077      562376.388      1868711.37      561387.308

Type RM Length L Ch R = 1 ,27000.5 ,259.2,261.8,264.4
XS GIS Cut Line= 4
     1882857.668      575502.744     1882347.392      575702.138
     1882105.767      575782.323     1881667.836       575850.57
#Sta/Elev= 30
       0  920.14    48.9  908.29   107.6  896.09   117.4  892.72   146.8   878.6
   264.1  818.59   303.3  799.94   332.6  786.79     362   774.3   381.5  767.17
   440.2  749.98   469.6   739.9   479.4  737.09   489.2  735.43   498.9  734.64
   596.8  727.86   659.8   725.4   675.1  725.03  687.83  725.79   694.7  727.13
   733.9  738.73   763.3  750.14   821.7  769.64   860.2  784.98   908.4  807.31
   985.5  841.25  1033.7  863.72  1091.5  893.02  1187.8  944.22  1245.6  972.38
#Mann= 3 , 0 , 0
       0     .08       0   659.8    .045       0  687.83      .1       0
Bank Sta=659.8,687.83
XS Rating Curve= 0 ,0
Exp/Cntr=0.3,0.1

Type RM Length L Ch R = 1 ,26738.6 ,233.1,214.8,196.6
XS GIS Cut Line= 4
     1882671.239      575374.285     1882405.142      575445.244
     1882032.607      575533.943     1881667.675      575713.875
#Sta/Elev= 30
       0  898.76    19.7  891.73    29.5  887.45    49.2  877.11    78.7  857.68
   127.9  820.51   147.5  806.56     177  788.68   196.7  779.08   206.6  775.05
   226.2  767.99   275.4  748.26   324.5  730.36   334.3  728.65   344.1  727.94
   449.4  722.52     462  722.03   471.8  722.64  475.67  723.68   481.6  725.25
   579.8  766.94   589.6  770.12     668  791.07   687.4  798.12   697.1  802.36
   764.9  834.65   813.4  858.83   929.6  921.88   958.7  937.04  1065.2  988.27
#Mann= 3 , 0 , 0
       0     .08       0   449.4    .045       0  475.67      .1       0
Bank Sta=449.4,475.67
XS Rating Curve= 0 ,0
Exp/Cntr=0.3,0.1

Type RM Length L Ch R = 1 ,26523.8 ,309,311.7,314.4
XS GIS Cut Line= 4
      1882502.53      574974.385     1882211.434       575189.13
     1882006.159      575417.213     1881641.167      575664.417
#Sta/Elev= 30
       0  871.33    68.4  840.98     176  800.59   224.9  783.75   303.1  759.09
   322.6  753.59     352  741.74   380.9  731.32   390.5  728.82   400.1  727.77
   428.9  726.77   505.6  721.79   541.3  720.39   553.5  720.22   563.1  720.88
   571.3  722.21   582.3  725.32   591.9  729.81     659  770.11   668.6  774.72
   678.4   778.6   727.4  796.78   776.4  820.82   835.1  852.68   952.7  920.38
   991.9  944.05  1011.5  955.14    1031  965.24  1050.6  974.58  1109.4 1000.56
#Mann= 3 , 0 , 0
       0     .08       0   541.3    .045       0   571.3      .1       0
Bank Sta=541.3,571.3
XS Rating Curve= 0 ,0
Exp/Cntr=0.3,0.1

Type RM Length L Ch R = 1 ,26212.1 ,213.6,213,212.4
XS GIS Cut Line= 2
     1882207.471       574799.01     1881553.633      575409.765
#Sta/Elev= 30
       0  873.35    19.7  862.62    39.3  852.57    68.8  838.98    98.3     826
   137.6  809.28   216.3  778.15   275.3  753.38   334.3  732.95   344.1   730.1
   363.8  725.56   398.8  720.71     413   719.6   422.8   719.9   428.8  720.52
   481.8  726.25   491.6  728.62   521.1  739.72   550.6  752.32   570.3  761.65
   589.9  771.54   629.2   792.6   678.4   820.6   757.1  867.08   766.9  872.51
   776.7   876.7   786.6  879.66   806.2  883.63   835.7   888.5   894.7  897.05
#Mann= 3 , 0 , 0
       0      .1       0   398.8    .045       0   428.8      .1       0
Bank Sta=398.8,428.8
XS Rating Curve= 0 ,0
Exp/Cntr=0.3,0.1

Type RM Length L Ch R = 1 ,25999   ,220.4,221.8,223.3
XS GIS Cut Line= 3
     1882173.737       574628.32     1881873.005      574817.545
      1881345.88      575331.154
#Sta/Elev= 30
       0   931.7    19.2  921.67    38.4  912.51    86.4   893.4   201.7  849.14
   240.1  833.32   278.5  815.94   345.7  782.51   355.3  777.06   433.8  727.97
   443.6  723.12   453.4  719.88   463.2  717.53   473.1  716.23   505.3  716.75
   523.6  715.94   535.3  717.07   610.4  722.47   620.3   724.2   630.1  727.93
   679.1   754.6   698.8  762.43     738   771.5   836.2  790.33   944.1   815.6
   963.7  819.24  1012.8   826.2  1032.4   831.5  1071.7  846.29  1091.3  852.76
#Mann= 3 , 0 , 0
       0     .08       0   505.3    .045       0   535.3      .1       0
Bank Sta=505.3,535.3
XS Rating Curve= 0 ,0
Exp/Cntr=0.3,0.1

Type RM Length L Ch R = 1 ,25776.9 ,264.5,281,297.4
XS GIS Cut Line= 3
     1882075.689      574545.584      1881599.25       574799.01
     1881274.865      575080.312
#Sta/Elev= 30
       0  940.64    39.2  924.04    49.1  920.34    78.5  911.17    88.3  907.46
   117.7  894.32   147.2  879.43   255.1  818.66   264.9  812.59   284.5  799.23
   323.8  770.25   353.2   749.8   372.8  737.83   402.3  721.92   412.1  718.18
   421.9  716.28   441.5  715.08   480.8   715.4   539.6  716.78   559.2  716.63
   568.7  715.96   588.4  713.75   598.7  713.84     608  715.48   627.5  722.31
   695.8  743.03   734.8  753.42   754.3  759.41   812.9   775.4     969  821.07
#Mann= 3 , 0 , 0
       0     .08       0   568.7    .045       0   598.7      .1       0
Bank Sta=568.7,598.7
XS Rating Curve= 0 ,0
Exp/Cntr=0.3,0.1

Type RM Length L Ch R = 1 ,25495.9 ,491.8,488.5,485.1
XS GIS Cut Line= 3
     1882062.235      574366.162     1881693.918       574526.95
     1881001.222      574645.215
#Sta/Elev= 30
       0  982.41    88.2   937.8   107.8  927.08   205.8  868.97   294.1  819.36
   333.3  795.92   431.2  739.14   460.4   721.3   470.2  716.84     480  714.36
   489.7  713.05   550.5  710.11   567.8   709.4   577.6  709.78   580.5  710.49
   587.3  712.16   597.1  716.79   616.6  727.66   626.4  733.57   675.2  766.24
   704.4  783.74   753.2  811.88     802  838.56   850.8  862.99   880.1  876.45
   919.2  893.55   948.4  905.69   977.7  917.02  1026.5  934.16  1104.6  959.12
#Mann= 3 , 0 , 0
       0      .1       0   550.5    .045       0   580.5      .1       0
Bank Sta=550.5,580.5
XS Rating Curve= 0 ,0
Exp/Cntr=0.3,0.1

Type RM Length L Ch R = 1 ,25007.4 ,360.7,368.8,376.9
XS GIS Cut Line= 3
     1881938.747        573904.6     1881558.702      574071.679
     1880922.604      574251.611
#Sta/Elev= 30
       0  968.36      29  955.08    96.6  921.86   173.8  885.16   299.3  822.63
     309  817.55   318.6  811.98   357.2  788.76   386.2  771.92     454  734.83
   473.5  726.08   502.6  714.38   512.4  710.96   531.8  706.13   542.7  704.32
   551.2  703.52     561  703.57   572.7  704.86   619.3  711.71     629  714.83
   648.5  723.74   677.6  737.93   716.5  759.03   784.6  794.74   823.4  816.23
   862.3  834.76   901.2  851.69   930.4  863.69   988.7   885.7  1076.2  920.66
#Mann= 3 , 0 , 0
       0      .1       0   542.7    .045       0   572.7      .1       0
Bank Sta=542.7,572.7
XS Rating Curve= 0 ,0
Exp/Cntr=0.3,0.1

Type RM Length L Ch R = 1 ,24638.5 ,449.1,441,432.9
XS GIS Cut Line= 3
     1881852.731      573753.158     1881163.414      573756.537
     1880788.344      573844.391
#Sta/Elev= 30
       0  942.14   116.5  874.43   145.6  858.48   223.3  822.54   252.4  807.68
   330.1  779.46   349.5  768.75   398.1  737.07   417.5  726.34     466  708.55
   475.7  706.07   495.1  703.68   504.9  703.33   525.1   704.5   592.2   710.6
   611.6  713.93   640.8  722.18   669.9  732.69     699  744.89   727.8  758.65
   756.7  774.87     853  837.97   891.6  861.48   930.1  882.24   968.6  900.04
   978.2  902.95   987.9  904.03   997.5  903.76    1036  900.92  1074.6   896.8
#Mann= 3 , 0 , 0
       0      .1       0   495.1    .045       0   525.1      .1       0
Bank Sta=495.1,525.1
XS Rating Curve= 0 ,0
Exp/Cntr=0.3,0.1

Type RM Length L Ch R = 1 ,24197.4 ,408.3,416.3,424.3
XS GIS Cut Line= 3
     1881819.507      573173.616     1881105.971      573374.709
     1880761.312      573648.409
#Sta/Elev= 30
       0  817.84   146.3  846.91   165.8  849.86   175.6  850.35   185.3   849.1
   224.4  835.81   390.2   774.5   409.7  764.62   458.5  735.77   487.7  719.39
   507.2  709.76   526.7  703.46   536.5  702.17   546.2  702.01   565.8   702.9
   643.8  709.88   663.3  712.62   692.6   721.5   760.9  747.17   780.4  752.16
     800  753.52   839.1  754.42   858.7  756.26   976.1  773.58  1005.4  781.94
  1054.3  798.32    1113  812.28  1122.8  813.83  1142.3  815.11  1181.4  813.92
#Mann= 3 , 0 , 0
       0      .1       0   526.7    .045       0   565.8     .08       0
Bank Sta=526.7,565.8
XS Rating Curve= 0 ,0
Exp/Cntr=0.3,0.1

Type RM Length L Ch R = 1 ,23781.1 ,348.9,337.1,326.1
XS GIS Cut Line= 3
     1881849.352      573104.389     1881393.186      572915.165
     1880664.021      572923.698
#Sta/Elev= 30
       0  782.39    87.2  777.05     184  775.14   242.1  775.72   300.2  772.33
   338.9  766.86     368  759.26   406.7  747.07   464.8  722.37   493.9  713.73
     523  709.05   552.2  706.28     630  704.88   660.8  702.41   678.6  701.41
   690.8  701.97   795.3   727.5     805  731.22   814.7  736.68   853.6  763.73
   863.3  767.72   882.8  770.49   902.2  774.77   950.8  789.96  1028.6  827.17
    1087  852.89  1125.8  867.98    1155  877.02  1174.5  881.84  1223.1  882.92
#Mann= 3 , 0 , 0
       0      .1       0   660.8    .045       0   690.8      .1       0
Bank Sta=660.8,690.8
XS Rating Curve= 0 ,0
Exp/Cntr=0.3,0.1

Type RM Length L Ch R = 1 ,23443.6 ,460.7,439.8,416.4
XS GIS Cut Line= 3
     1881859.489      572323.839      1881413.46      572496.168
     1880647.666      572811.352
#Sta/Elev= 30
       0  887.68     9.8  883.72      39  867.04    87.8  852.78   146.4  824.73
   165.9   817.4   185.4  811.72   253.7  795.45   361.1  776.74   419.6  761.97
   517.1  733.86   653.5  702.96     728  696.45   741.2     696     758  697.86
   789.9  704.34   848.4  726.38   867.9  735.86   916.6  765.73   936.1  774.29
   945.8  777.33   984.8  785.55  1004.3  792.08  1023.8  800.11    1053  815.81
  1111.4  851.83  1130.9  862.12  1150.4  870.81  1179.6  880.01  1306.3   912.2
#Mann= 3 , 0 , 0
       0      .1       0     728    .045       0     758      .1       0
Bank Sta=728,758
XS Rating Curve= 0 ,0
Exp/Cntr=0.3,0.1

Type RM Length L Ch R = 1 ,23003.7 ,541.6,553.4,565
XS GIS Cut Line= 3
     1881160.035        571911.6     1880920.126      572472.515
     1880576.354      572736.446
#Sta/Elev= 30
       0  838.69    29.5  825.04      59  812.68    98.4  799.35   137.8  785.38
   157.4  779.03   216.5  762.57   334.6  727.65   413.3  702.82   423.1   700.2
     433  698.37   462.8  694.99   482.2  694.32   492.8  695.08   521.5  699.59
   560.9  703.04   570.7   705.4   580.6  709.26   619.7  727.49     639  737.15
     716   777.8   744.9  791.95   783.4   813.4   793.1  818.39   831.6   836.7
   879.7  858.61   908.6  871.06   956.8   889.7   995.3  903.07  1043.5   918.2
#Mann= 3 , 0 , 0
       0      .1       0   462.8    .045       0   492.8      .1       0
Bank Sta=462.8,492.8
XS Rating Curve= 0 ,0
Exp/Cntr=0.3,0.1

Type RM Length L Ch R = 1 ,22450   ,319.8,320.7,322.8
XS GIS Cut Line= 3
     1880939.724      571634.313        1880551.      572017.753
     1880164.912      572403.821
#Sta/Elev= 30
       0   862.1    48.8  833.24    58.5  828.44   107.2  809.67     117  806.27
   136.5  801.12   243.8  776.85   263.3  771.79   302.3  758.41     351  739.69
   360.8   736.5     468  709.99   497.3  703.22   530.9   696.1   536.3  694.94
     546  693.64   555.8  693.46   560.9  694.23   565.5  694.93   594.8  702.47
   604.5  705.18   614.3   708.9     624  713.82   721.5  765.84     741   775.4
   828.8  812.93     858  824.87   984.8  872.58    1014  885.32    1092  918.49
#Mann= 3 , 0 , 0
       0      .1       0   530.9    .045       0   560.9      .1       0
Bank Sta=530.9,560.9
XS Rating Curve= 0 ,0
Exp/Cntr=0.3,0.1

Type RM Length L Ch R = 1 ,22129.2 ,461.1,452,443
XS GIS Cut Line= 2
     1880709.727      571458.863     1879997.601      572079.755
#Sta/Elev= 30
       0     849    29.5  831.96    49.2  821.32      59  816.97    68.9  813.24
    88.6  808.26   216.5  781.73     246  774.85   255.9  771.61   275.6  763.73
   324.8  742.32   423.2  700.78     433  696.91   442.9  694.08   452.7  692.94
   462.6  692.78   472.4  692.98   570.8  696.93   590.5  698.23   610.2   702.1
   649.5  712.62   659.4  714.68   688.9  718.76   698.8  721.16   718.4   728.6
     748  741.31   777.5  754.84   826.7  778.84   846.4  787.41   944.8  819.74
#Mann= 3 , 0 , 0
       0      .1       0   442.9    .045       0   472.4     .06       0
Bank Sta=442.9,472.4
XS Rating Curve= 0 ,0
Exp/Cntr=0.3,0.1

Type RM Length L Ch R = 1 ,21677   ,490.3,521.5,552.7
XS GIS Cut Line= 3
     1880505.878      571133.393     1880065.237      571414.886
     1879686.789      572026.486
#Sta/Elev= 30
       0  909.05    87.2  893.94   135.6  881.16   154.9  874.68     213  852.96
   300.2  815.72   406.7  776.64     426  768.49   455.1  755.34   464.8  751.62
   513.2  737.74   532.6  731.01   590.9  704.43   600.6  700.65   610.4  697.55
   629.8  692.78   639.5  690.74   649.2  689.91     659  690.59     795  704.73
   853.3  710.08   872.8  713.82   901.9  721.26   921.4  727.28   999.1  754.35
  1018.6  758.88  1057.4  766.81  1183.8   790.5  1203.2  792.02  1242.1   791.5
#Mann= 3 , 0 , 0
       0      .1       0   629.8    .045       0     659     .06       0
Bank Sta=629.8,659
XS Rating Curve= 0 ,0
Exp/Cntr=0.3,0.1

Type RM Length L Ch R = 1 ,21155.4 ,730.4,869.8,758.8
XS GIS Cut Line= 3
     1880436.278      571056.405     1880076.163      571101.533
     1879113.147      571114.204
#Sta/Elev= 30
       0  871.37    39.2  859.81    88.3     844   137.3  835.31   166.8  828.08
   186.4  822.33   264.8  797.07   294.3  784.25   421.9  725.28   490.7  695.63
   500.5  692.87   510.3  691.64     645  688.01   657.8  687.63   667.6  687.79
     675  688.74   726.6  701.82   746.2  708.15   775.7  718.86   844.5  746.88
   923.1  780.84  1011.6  821.03  1109.8  868.45    1159  893.72  1217.9  927.43
  1237.6  937.57  1247.4  941.25  1257.2  943.56  1296.6  948.05    1326  953.12
#Mann= 3 , 0 , 0
       0     .08       0     645    .045       0     675      .1       0
Bank Sta=645,675
XS Rating Curve= 0 ,0
Exp/Cntr=0.3,0.1

Type RM Length L Ch R = 1 ,20284.6 ,546.7,549.4,552.4
XS GIS Cut Line= 3
     1880406.351      570790.073      1879894.88      570549.547
     1879357.019      570347.325
#Sta/Elev= 30
       0  820.55    29.2  813.62    58.5  803.98   107.2  784.99   126.7  772.48
   136.4  767.47   175.4  756.09   204.6  745.74   263.1  731.54   311.8  716.77
   360.6  703.96   448.3  686.58     458  685.11   467.8  684.91   477.5  685.79
     497  689.96   565.2  697.09   604.2  697.79   613.9  700.86   633.4  713.04
   652.9  723.27   672.3   730.3   701.6   738.6     760  746.06   789.2  751.22
   886.6   778.6   974.3  796.84    1023  808.42  1071.6  815.96  1139.8     820
#Mann= 3 , 0 , 0
       0      .1       0   448.3    .045       0   477.5      .1       0
Bank Sta=448.3,477.5
XS Rating Curve= 0 ,0
Exp/Cntr=0.3,0.1

Type RM Length L Ch R = 1 ,19734.3 ,392.2,386.1,379.6
XS GIS Cut Line= 3
     1880697.111      570489.039     1880433.549      570330.226
     1879736.177      569881.779
#Sta/Elev= 30
       0  844.66    57.7   841.4    86.5  838.46   115.4  833.36   134.6  828.93
   153.9  823.34   230.8  795.06     337  749.43   356.5  740.07   444.3  694.11
     454  690.17   463.8  688.19   502.9   684.8   522.3   683.1   541.8  685.02
   629.6  702.81   668.6  713.93   688.1  716.05   736.9  718.41   746.7  719.91
   766.2  726.23   795.4  732.96   814.9  739.94   844.2  752.08   863.7  758.54
   922.2  772.34   980.8  783.18  1019.8  794.02  1088.1  815.54  1136.8  836.28
#Mann= 3 , 0 , 0
       0      .1       0   502.9    .045       0   541.8      .1       0
Bank Sta=502.9,541.8
XS Rating Curve= 0 ,0
Exp/Cntr=0.3,0.1

Type RM Length L Ch R = 1 ,19348.2 ,454.2,427.1,399.8
XS GIS Cut Line= 3
     1880886.741      570066.196     1880156.471      569816.617
     1879775.076      569784.135
#Sta/Elev= 30
       0  765.68    58.6  752.22   107.5  742.31   195.4  729.91     254  724.68
   293.1  720.07   371.2  706.78   449.4  691.65   468.9  689.66   556.8  685.23
   575.7  683.44   586.1  682.19   595.9  682.38  600.74  683.54   605.7  684.69
     635  696.17   654.5  702.22   703.4  715.48   742.4  724.79     762  728.79
   801.2  732.62   830.6  741.97   860.1  748.84   899.3  755.48   948.4  761.31
   987.7  769.54  1046.6  786.26    1076  795.44  1115.3  808.86  1154.5  823.41
#Mann= 3 , 0 , 0
       0     .08       0   575.7    .045       0  600.74     .08       0
Bank Sta=575.7,600.74
XS Rating Curve= 0 ,0
Exp/Cntr=0.3,0.1

Type RM Length L Ch R = 1 ,18921   ,421.3,431.2,441.2
XS GIS Cut Line= 3
     1880799.503      569284.209     1880119.301      569651.046
     1879767.809      569691.906
#Sta/Elev= 30
       0  825.51    68.5  828.75     137  830.83   146.7  830.45   156.5  829.04
   166.3  826.39   244.6  801.64   264.1  794.15   293.5  780.47   332.6  763.28
   342.4  758.39   430.4   710.5   440.2  705.42     450  701.15   469.6  695.65
   528.2  682.14     538  680.45   547.8  680.08     565  682.82   596.7  686.21
   645.6  692.72   684.8  701.74   733.7  711.59   792.5  719.95     822  725.96
   861.3  736.47   939.9  761.56  1018.6  785.51  1067.7  801.83  1126.7   822.8
#Mann= 3 , 0 , 0
       0      .1       0   528.2    .045       0     565     .06       0
Bank Sta=528.2,565
XS Rating Curve= 0 ,0
Exp/Cntr=0.3,0.1

Type RM Length L Ch R = 1 ,18489.7 ,484.6,484.8,485.1
XS GIS Cut Line= 3
     1880729.322      569107.183     1880322.042      569123.921
     1879551.629      569245.565
#Sta/Elev= 30
       0  749.31    67.9  743.56   126.2  735.65   184.4  732.06   271.8  730.66
   310.6  733.12     330  731.39   427.1  713.06   446.6  706.44   485.6  690.17
   531.8  678.78   544.1  677.86   561.8   679.3   670.9  681.19   680.6  682.22
   748.9  697.46   836.6   730.9   875.6  743.44   914.6  753.58   953.6  761.47
   982.8  765.78  1002.3  765.74  1031.6   759.9  1041.3  760.27  1060.8  763.91
  1080.3  765.04  1109.6   769.2  1129.1  772.54  1148.6   778.4  1187.6  796.83
#Mann= 3 , 0 , 0
       0     .08       0   531.8    .045       0   561.8     .08       0
Bank Sta=531.8,561.8
XS Rating Curve= 0 ,0
Exp/Cntr=0.3,0.1

Type RM Length L Ch R = 1 ,18004.6 ,461.8,457.4,453.1
XS GIS Cut Line= 3
     1880653.184      568633.965     1880271.357       568684.65
     1879487.427      568796.157
#Sta/Elev= 30
       0   826.7    38.5   823.7    86.7  818.18   125.2  811.92   154.1  803.88
   231.1  778.95   269.6   765.5   298.5  753.34   365.9  722.44   424.3  694.23
     434  690.17   443.8  687.45   463.4     685   492.7  682.63   551.4  680.36
   619.8  676.72   639.3  675.86   649.1  676.63   658.9  679.32   668.7  682.81
   678.4   685.3     698   689.2   707.8  692.21   717.6   695.9   737.1  704.22
     786  726.28   883.7  765.46   952.2  791.17  1020.6  813.48    1177  866.37
#Mann= 3 , 0 , 0
       0     .06       0   619.8    .045       0   649.1      .1       0
Bank Sta=619.8,649.1
XS Rating Curve= 0 ,0
Exp/Cntr=0.3,0.1

Type RM Length L Ch R = 1 ,17547.1 ,365.1,361,357
XS GIS Cut Line= 4
     1880504.508      568204.831     1880162.328      568222.621
     1879798.477       568334.26     1879497.564      568458.257
#Sta/Elev= 30
       0  857.52      49  846.86    88.1  839.91   107.7  834.81   117.5  831.36
   137.1  822.54   166.4   807.1   205.6  787.84   264.3  761.35   313.3  741.36
   352.4  729.02   371.9  721.84   430.5  698.56   459.8  685.69   485.9  675.43
     489   674.3   498.8  672.55   515.9  673.73   537.8  675.83   645.2  682.13
   674.4  686.51   684.2   688.5     694  691.37   713.5  699.88   761.5  723.53
   790.2  736.13   905.1  788.82   962.5  812.24  1010.4  829.39  1048.7  844.16
#Mann= 3 , 0 , 0
       0     .08       0   485.9    .045       0   515.9     .06       0
Bank Sta=485.9,515.9
XS Rating Curve= 0 ,0
Exp/Cntr=0.3,0.1

Type RM Length L Ch R = 1 ,17186.1 ,691.7,663.8,635
XS GIS Cut Line= 4
     1880186.037      567538.323     1880016.265      567906.605
     1879626.255      568087.882     1879302.913      568317.368
#Sta/Elev= 30
       0  806.92    57.9  777.54    77.2  768.78   106.2  757.47   154.5  742.36
   299.3  703.25   337.9   696.8   405.5  688.22   434.8  686.11   483.7  684.73
     601  677.47   621.8  673.54   630.3  672.23   640.1  672.83   649.9   675.9
   659.7  680.26   669.4  683.53   698.8  684.13   737.9  691.97   796.5  715.94
   845.3  730.86   864.6   737.4   903.3  753.48     942  775.56    1087   839.8
  1106.4  847.68  1135.4  856.44  1154.8  863.31  1183.8  874.79  1232.1  895.58
#Mann= 3 , 0 , 0
       0     .06       0   621.8    .045       0   649.9     .08       0
Bank Sta=621.8,649.9
XS Rating Curve= 0 ,0
Exp/Cntr=0.3,0.1

Type RM Length L Ch R = 1 ,16522.2 ,420.8,349.1,391.5
XS GIS Cut Line= 3
     1879710.442      567113.413     1879450.258      567431.039
      1879223.04      568248.026
#Sta/Elev= 30
       0  826.71    97.8  817.16   166.2  806.29   185.7  802.26   205.3  795.34
   244.4  777.43   283.5  761.34   381.3   728.6   410.6   714.7   459.3  693.06
   488.6  681.12   498.3  678.66   508.1  677.38   576.3  672.76     599  670.09
   615.3  668.78     629  670.11     703   674.6   722.5  676.98     781  692.12
   829.7  708.47   868.7  720.23   966.2  751.97   995.4  762.49  1024.6  776.36
  1102.6   820.4  1131.9  838.45  1151.4  848.07  1180.6  859.69  1258.6  884.53
#Mann= 3 , 0 , 0
       0     .06       0     599    .045       0     629     .06       0
Bank Sta=599,629
XS Rating Curve= 0 ,0
Exp/Cntr=0.3,0.1

Type RM Length L Ch R = 1 ,16172.6 ,577.1,566.3,555.5
XS GIS Cut Line= 3
     1879007.609       566917.43      1879038.02      567319.532
     1879115.138       568235.14
#Sta/Elev= 30
       0  829.79    68.8  813.59    88.5  804.38   147.5  770.15   167.2  760.71
   186.9  752.85   226.2  740.82   383.6  698.58   403.2  694.47   452.1  686.97
   510.8  675.12   628.1  670.96   643.1  669.31   657.4  667.69   673.1  668.88
   686.7  670.22   755.2  671.59   774.7  672.94   823.6  685.25   921.3  724.52
   970.2  740.69  1009.3  755.82  1048.4  773.73  1087.5  797.41    1107  805.68
  1146.2  820.03  1175.5  829.76  1263.4  855.62  1292.8   862.4  1322.1  866.65
#Mann= 3 , 0 , 0
       0     .06       0   643.1    .045       0   673.1     .06       0
Bank Sta=643.1,673.1
XS Rating Curve= 0 ,0
Exp/Cntr=0.3,0.1

Type RM Length L Ch R = 1 ,15606.5 ,547.7,559.9,571.7
XS GIS Cut Line= 3
     1878429.799       567191.13     1878811.626      567991.954
     1878919.755      568225.105
#Sta/Elev= 30
       0  851.03    58.5  828.05      78  821.52     117  812.52     156  809.13
   175.5  804.55     195  798.47   214.5  789.99     273  759.21   302.2  746.82
   341.2  732.38   409.5   708.6   477.7  688.04   516.7   677.9     546  671.63
   594.7  668.94     663  669.12   689.7  665.29     702  664.48   711.7  665.43
   719.7  667.57   750.7  676.19   760.4  680.25     858  724.42   944.3  765.55
   991.9  786.36  1020.4  797.71    1049  805.57    1068  808.71  1144.2  813.13
#Mann= 3 , 0 , 0
       0      .1       0   689.7    .045       0   719.7      .1       0
Bank Sta=689.7,719.7
XS Rating Curve= 0 ,0
Exp/Cntr=0.3,0.1

Type RM Length L Ch R = 1 ,15045.9 ,592.8,591.2,589.6
XS GIS Cut Line= 3
     1878169.615      567285.742     1878206.784      567691.223
     1878233.817      568468.394
#Sta/Elev= 30
       0  873.68      97  838.66   184.2  803.96   261.8  769.47   329.6     738
   465.5  678.92   494.7  668.85   504.4   666.3   519.5  663.56   533.6  662.86
   549.5  664.34   572.4  665.26     621  663.97   640.5  664.18   669.6     666
   679.4   667.4   689.1  669.68     728  683.16   766.8  695.27   786.3     704
   834.9  729.79   854.3  738.65  1029.3  804.33  1048.7  810.38  1058.5  812.31
  1077.9  814.96  1107.1  817.11  1116.8   818.5  1126.5  821.01  1184.8  839.98
#Mann= 3 , 0 , 0
       0      .1       0   519.5    .045       0   549.5     .08       0
Bank Sta=519.5,549.5
XS Rating Curve= 0 ,0
Exp/Cntr=0.3,0.1

Type RM Length L Ch R = 1 ,14454.6 ,318.9,336.8,354.6
XS GIS Cut Line= 3
     1877726.966      567353.322     1877618.838      567725.013
     1877696.555      568590.038
#Sta/Elev= 30
       0  834.91    58.1  825.84    77.4   821.9   106.4  814.81   222.6  778.53
   280.6   757.4   377.4   732.7   387.1  728.68   396.9  722.14   406.6  714.04
   455.4  670.47   465.2  663.66   474.9  660.93   494.4  662.85   640.8  670.84
   670.1  673.59   679.8  676.26   689.6  680.13   728.6  696.92   748.2  707.38
   787.2  732.18     797  737.69   806.7  742.07   914.1  779.33   943.3  788.82
   962.8  794.05  1011.6   804.1  1070.2  817.82  1138.5  832.49  1255.6  854.84
#Mann= 3 , 0 , 0
       0      .1       0   465.2    .045       0   494.4     .06       0
Bank Sta=465.2,494.4
XS Rating Curve= 0 ,0
Exp/Cntr=0.3,0.1

Type RM Length L Ch R = 1 ,14117.8 ,542.9,573.9,605
XS GIS Cut Line= 3
     1877686.418      567339.806     1877402.581      567583.094
     1876990.343      568323.097
#Sta/Elev= 30
       0  841.45    39.4  840.78      59  839.25    78.7  833.32    98.4  824.13
   127.9   805.8   147.6  795.64   186.9  778.69   226.3  764.84   295.1   735.1
     305  731.78   334.5  725.12     403  703.53   422.5  696.43     442  687.71
   461.5  673.47   471.2  667.92   510.2  661.44   519.9  660.43   539.4  661.34
   607.5  666.09   665.9  672.66   753.6  679.58   841.2  689.37   919.1  701.93
   987.2  721.62  1045.7  734.42    1182  758.86  1201.4  760.45  1220.9     760
#Mann= 3 , 0 , 0
       0      .1       0   510.2    .045       0   539.4     .08       0
Bank Sta=510.2,539.4
XS Rating Curve= 0 ,0
Exp/Cntr=0.3,0.1

Type RM Length L Ch R = 1 ,13543.8 ,523,501.6,480.3
XS GIS Cut Line= 3
     1877723.587      567126.929     1877358.654       567191.13
     1876621.169      567215.573
#Sta/Elev= 30
       0  855.67    29.2   852.3      78  842.34    97.5  835.33   146.3  814.67
     195  798.98   243.8  773.41   321.8  725.42   380.4  694.65     400  685.25
   449.2  665.92   459.1   662.6   468.9  660.95   518.1  660.64   537.8  659.36
   547.6  658.48   567.3  661.01   655.8  679.62   675.5  689.33   714.9  715.31
   724.7  720.87   734.6  724.66   783.8  732.03   813.3  738.02   842.8  745.32
   862.5  751.72   901.8  769.23   970.7  807.21  1000.2   822.3  1108.4  869.54
#Mann= 3 , 0 , 0
       0     .08       0   537.8    .045       0   567.3      .1       0
Bank Sta=537.8,567.3
XS Rating Curve= 0 ,0
Exp/Cntr=0.3,0.1

Type RM Length L Ch R = 1 ,13042.1 ,340.8,337.8,334.8
XS GIS Cut Line= 4
      1877470.95      566347.273     1877176.977      566610.835
     1876961.565      566800.904     1876562.984      567120.209
#Sta/Elev= 30
       0  797.49    28.9  789.71   134.8  751.56   154.1  745.73   231.1  725.98
   288.9  705.08   308.2  701.88   327.4   703.2   356.3   708.5   365.9  708.84
   385.2  706.27   442.7  695.28   452.3  690.94   471.4  677.94     481   673.6
   528.9  665.87   566.7  656.93   576.8  656.26   596.7  658.39   643.8  665.02
   691.9  668.48   711.6  673.92   770.5  694.95   888.4     748   947.3  775.66
   976.7  791.22  1045.5  813.63  1065.1  821.39  1163.3  869.32  1192.8  882.46
#Mann= 3 , 0 , 0
       0     .08       0   566.7    .045       0   596.7     .08       0
Bank Sta=566.7,596.7
XS Rating Curve= 0 ,0
Exp/Cntr=0.3,0.1

Type RM Length L Ch R = 1 ,12704.3 ,223.8,224.8,225.8
XS GIS Cut Line= 3
      1877214.99      566291.519     1876844.989      566496.794
     1876429.372      566945.357
#Sta/Elev= 30
       0  756.24   108.2  739.47     187  730.26   226.3  724.67   314.9  715.66
   354.2  710.98   364.1  709.28   383.8  703.97   423.1  692.08   452.2  686.79
   491.1  676.79   520.2  668.26  553.72  656.82     559  655.23   568.7  653.76
   578.4  654.62  582.89  656.06   617.3  668.64   694.9   690.1   704.6  693.19
   714.3   697.1   801.7  743.43   879.3  789.54   898.8   802.2   947.3  839.61
   966.7  852.74   976.4  858.19   995.8  867.01  1015.2  874.34  1034.6  880.63
#Mann= 3 , 0 , 0
       0     .06       0  553.72    .045       0  582.89     .08       0
Bank Sta=553.72,582.89
XS Rating Curve= 0 ,0
Exp/Cntr=0.3,0.1

Type RM Length L Ch R = 1 ,12479.5 ,513.9,491.1,468.4
XS GIS Cut Line= 3
     1876987.823       565977.18     1876715.241      566317.627
      1876241.54      566796.106
#Sta/Elev= 30
       0   783.9    38.8  774.32    67.8  765.64    87.2  756.68   116.3  741.11
   135.7  729.19   145.4  724.92   184.1  717.46   213.2  706.63   232.6  701.32
   319.8  699.66   387.7  694.37   436.1  684.05   484.9  668.52   504.4  663.38
     524  660.41   553.2  658.23   571.5  655.16   592.2  652.63   601.5  653.66
   660.6  665.98   680.1  671.23   748.4  700.23   777.6  711.12   787.4     717
   875.2   777.2   894.8  788.54   904.5  792.11   982.6  805.07  1109.4   839.2
#Mann= 3 , 0 , 0
       0     .06       0   571.5    .045       0   601.5     .08       0
Bank Sta=571.5,601.5
XS Rating Curve= 0 ,0
Exp/Cntr=0.3,0.1

Type RM Length L Ch R = 1 ,11988.7 ,572.6,554.2,534.6
XS GIS Cut Line= 4
     1876246.021      565584.661     1876238.884      565829.685
     1876200.822      566348.282      1876115.18      566731.585
#Sta/Elev= 30
       0  685.32    19.6  681.77    29.4  680.57      98   674.1   147.1  674.02
   196.1  670.32   274.6  666.72   362.9   660.5     461  655.92   519.8  654.35
   551.4  651.95   559.1  651.61   568.9  651.86   581.4  653.19   588.5   654.1
     618  654.69   627.8  655.72   657.2  660.62     667  662.76   696.4  672.52
   755.3  688.47   804.4  703.51     824  710.74   833.8  715.04   873.1  733.34
   922.2  757.98   971.3  778.48  1030.2  798.89  1108.8  822.43  1157.9  839.74
#Mann= 3 , 0 , 0
       0     .06       0   551.4    .045       0   581.4     .06       0
Bank Sta=551.4,581.4
XS Rating Curve= 0 ,0
Exp/Cntr=0.3,0.1

Type RM Length L Ch R = 1 ,11434.1 ,318.6,320.1,323.8
XS GIS Cut Line= 3
     1875616.582      565935.321      1875882.73      566427.575
     1876037.463       566714.69
#Sta/Elev= 30
       0  806.28    49.1   790.6    88.4   774.1     108  764.18   157.1  734.08
   186.5  717.85     216  703.77   245.4  692.99   265.1  687.86   274.9  687.14
   353.4   685.1   363.2  682.91   382.9  673.82   392.7  670.53     432  660.43
   451.1  652.53   461.4  649.54   471.2  649.42   481.1  651.57   500.7  656.57
   520.3  660.37   569.2  667.73   588.4  672.98   607.6  680.47   626.8  689.42
   645.9  699.46   818.6  792.74   837.8  802.52   876.2  820.07   885.8   825.6
#Mann= 3 , 0 , 0
       0     .08       0   451.1    .045       0   481.1     .08       0
Bank Sta=451.1,481.1
XS Rating Curve= 0 ,0
Exp/Cntr=0.3,0.1

Type RM Length L Ch R = 1 ,11114   ,653.7,651.5,646.9
XS GIS Cut Line= 3
     1875319.181        565985.6     1875557.426      566476.884
     1875758.089      566988.162
#Sta/Elev= 30
       0  813.47    58.5  810.84      78   808.6   185.2  779.22   214.5  772.59
   224.2  769.06   243.8  757.98     273  743.61   370.5  689.97     429  660.35
   438.8  656.94   448.5  655.17     507  651.34   526.5   648.3   536.2  647.98
   555.8  651.04   614.7  662.08   653.9  670.97   702.9  679.59   712.7  683.24
   742.2  698.71   810.8  721.36   820.6  726.49   889.3  774.47   899.1  780.12
   908.9  783.73   938.3  789.97   967.8  798.91  1046.2  826.12  1095.2  840.08
#Mann= 3 , 0 , 0
       0     .06       0   526.5    .045       0   555.8     .06       0
Bank Sta=526.5,555.8
XS Rating Curve= 0 ,0
Exp/Cntr=0.3,0.1

Type RM Length L Ch R = 1 ,10462.4 ,771.2,794.9,818.6
XS GIS Cut Line= 3
     1874648.692      566234.871     1874908.875      566616.699
     1875310.977      567272.226
#Sta/Elev= 30
       0  885.87    19.7  882.24    78.6   867.4   127.8   861.1   147.5  857.14
   186.8  842.81   196.6  838.24   245.8  806.88   324.4  769.96   353.9  754.67
   373.6  743.01   442.4   698.1   471.8  681.62   520.4  659.92   549.7  652.77
   571.1  645.96   578.9     645   601.1  646.84   617.8  648.49   676.2  649.12
   695.7  650.62   724.9  656.61     793  674.92   822.2  685.54     939  745.09
   968.2  759.47   987.7  767.51  1046.1  779.57  1133.7  794.22  1231.1  821.68
#Mann= 3 , 0 , 0
       0      .1       0   571.1    .045       0   601.1     .08       0
Bank Sta=571.1,601.1
XS Rating Curve= 0 ,0
Exp/Cntr=0.3,0.1

Type RM Length L Ch R = 1 ,9667.1  ,613.4,619.8,625.8
XS GIS Cut Line= 4
     1874505.873       566494.26     1874551.489      567021.384
     1874447.585      567426.865     1874513.532      567941.269
#Sta/Elev= 30
       0  828.51    68.6  816.74   117.6  805.36     196  779.08   215.6  775.74
   225.4  771.56     245   759.6   254.8  755.01   264.6  752.21   323.3  740.18
   440.9  726.53   470.3  721.09   529.1  700.96   616.7  657.97   626.4  654.03
   636.2  651.96   710.4  644.18   723.8  642.99   740.4  644.07   811.4     652
   908.7  655.62   986.8  669.26  1065.1  694.25  1192.3  748.52  1211.9  754.92
  1260.8  765.26  1319.5  773.96  1397.8   796.1  1427.2  799.73  1466.3  801.43
#Mann= 3 , 0 , 0
       0     .06       0   710.4    .045       0   740.4     .06       0
Bank Sta=710.4,740.4
XS Rating Curve= 0 ,0
Exp/Cntr=0.3,0.1

Type RM Length L Ch R = 1 ,9046.8  ,651.9,637.3,623.3
XS GIS Cut Line= 3
     1874244.003      566491.463     1874165.494      566930.946
     1873816.556      567586.523
#Sta/Elev= 30
       0  833.36    77.6  816.78   203.8  792.81     262  775.62   300.9  758.16
   359.1  724.52   417.3  693.73   436.7  684.45   505.1  657.77   524.6  647.81
   534.4  644.25   559.5  642.51   573.5  641.54   589.5  642.73   602.8   644.4
   661.4  647.43   690.7  650.64   710.3  654.82   768.9  670.06     808   677.3
   817.8   680.4   827.5  684.81   886.2  717.92   905.7  727.82  1003.4  773.92
  1032.8  785.78  1071.8  799.01  1101.2  806.52    1150  816.39  1189.1  821.92
#Mann= 3 , 0 , 0
       0      .1       0   559.5    .045       0   589.5     .08       0
Bank Sta=559.5,589.5
XS Rating Curve= 0 ,0
Exp/Cntr=0.3,0.1

Type RM Length L Ch R = 1 ,8409.5  ,603.8,613.5,624.2
XS GIS Cut Line= 3
     1873543.757       566478.16     1873513.346      566907.293
      1873499.83      567586.474
#Sta/Elev= 30
       0  826.01    29.3  820.97    68.4  817.14    78.2  814.99    97.8  808.75
   107.6  806.45   166.2  794.88   215.1  787.65   224.9  784.99   283.6  759.07
   312.9  749.24   322.7   743.2   342.2  724.92     352  717.93   361.8  713.27
   410.6   693.6     469  664.35   546.7  642.38   556.4  640.02   575.8   639.2
   595.2  640.32   624.3  642.71   643.7  645.18   672.8   652.9   740.8  673.18
   779.6  689.23   934.8  758.41  1002.8  782.62  1070.7  809.06  1109.5  825.51
#Mann= 3 , 0 , 0
       0     .06       0   546.7    .045       0   595.2     .06       0
Bank Sta=546.7,595.2
XS Rating Curve= 0 ,0
Exp/Cntr=0.3,0.1

Type RM Length L Ch R = 1 ,7795.9  ,484.2,490.4,495.7
XS GIS Cut Line= 3
     1873259.921      566315.968     1873040.285      566674.142
     1872776.723      567333.048
#Sta/Elev= 30
       0  843.23    78.2   829.1   107.5  820.53     127  812.76   146.6   803.8
   185.6  784.24   244.3  756.16   322.4  715.09   381.1  682.25   410.4  668.22
   429.9  661.36     459  653.94   478.5  650.21   527.1  643.11   543.3  640.09
   556.2  639.11   573.3  639.91   624.3  647.17   692.4   659.1   702.1   661.6
   711.8   665.5   877.1  742.52   925.7  766.08     984  796.48   993.7  800.19
  1003.4  802.44  1032.6  807.25    1052  809.56  1081.2  810.72  1129.8  810.61
#Mann= 3 , 0 , 0
       0      .1       0   543.3    .045       0   573.3     .06       0
Bank Sta=543.3,573.3
XS Rating Curve= 0 ,0
Exp/Cntr=0.3,0.1

Type RM Length L Ch R = 1 ,7305.4  ,407.8,429.7,451.5
XS GIS Cut Line= 3
     1872793.618      566234.871     1872472.613      566768.754
     1872056.995      567069.486
#Sta/Elev= 30
       0  804.25    68.1  779.55    87.6  774.29   155.7  758.91   165.5  755.59
   243.3  715.42   311.5  685.44   369.9   657.5   379.6  653.64   399.1  648.74
     438  642.62   457.9  638.08   467.2  636.72     477  637.25   487.9  639.75
   496.4  641.98   515.9  643.52   632.6  645.96     681  648.76   739.1  655.99
   758.5  661.29   777.8  668.06   787.5  672.28   816.5  687.12   864.9  714.67
   932.7  756.61  1019.8  807.06  1039.2  816.19  1058.5  824.19    1136  850.65
#Mann= 3 , 0 , 0
       0     .06       0   457.9    .045       0   487.9     .06       0
Bank Sta=457.9,487.9
XS Rating Curve= 0 ,0
Exp/Cntr=0.3,0.1

Type RM Length L Ch R = 1 ,6875.6  ,373.8,377,380.4
XS GIS Cut Line= 3
     1872803.755      566201.081     1872161.744      566397.064
      1871698.82       566613.32
#Sta/Elev= 30
       0  815.62    97.3  779.56   126.5  770.12   155.6  761.99   165.4  757.94
   291.8  689.91   369.7  654.41   389.1  649.85   447.5   642.8   486.4  639.78
   544.8  637.69     574  634.22   583.7   634.1   593.4  635.42   603.2  638.46
   632.3  647.22   720.4   666.9   730.2  669.82     740   673.7   789.2  697.38
     858  736.04   867.8  739.22   907.1  745.05   956.2  756.68   975.9  762.55
    1025  779.57  1103.6  799.57  1123.2  807.04  1152.7  822.06  1182.2  832.34
#Mann= 3 , 0 , 0
       0     .06       0     574    .045       0   603.2     .06       0
Bank Sta=574,603.2
XS Rating Curve= 0 ,0
Exp/Cntr=0.3,0.1

Type RM Length L Ch R = 1 ,6498.6  ,245.2,258.6,271.8
XS GIS Cut Line= 3
     1872695.865      565903.532      1872126.47      566012.955
     1871594.329      566105.454
#Sta/Elev= 30
       0   828.8    49.1   806.5    78.6  794.72   137.6  780.32   196.6  759.85
   216.2   751.9   245.7  738.21     285  717.84   304.6  705.64   334.1  685.82
   353.8   674.8   393.1  656.46   422.6  644.96   432.4  642.24   442.2  640.82
   520.8  637.69   530.7     637   544.9  634.56   560.2  632.66   574.9  635.23
   599.4  640.92   736.9  663.16   756.6  667.71   776.2   674.9   795.9  683.59
   805.7  688.28     845  709.71   933.4  751.04  1051.2  786.55  1119.9   805.3
#Mann= 3 , 0 , 0
       0     .06       0   544.9    .045       0   574.9     .06       0
Bank Sta=544.9,574.9
XS Rating Curve= 0 ,0
Exp/Cntr=0.3,0.1

Type RM Length L Ch R = 1 ,6240.2  ,509.2,489.5,469.9
XS GIS Cut Line= 4
     1872729.417      565815.875     1872373.323      565809.105
     1872024.838      565718.778     1871681.925      565677.336
#Sta/Elev= 30
       0  839.41    38.5  823.84   105.9  795.37   134.8  783.83   240.6  735.46
   250.3  730.55   259.9  725.13   336.9  679.35   346.5  674.02   356.2  669.52
   375.6  662.46     434  642.89   443.7  641.04   453.5  640.42   492.4   639.5
   511.8  638.56   521.6  637.42     533  634.86     541  633.01   550.8  632.51
     563   634.7   579.9  639.34   677.2  664.07     687  667.48   696.7  671.89
   783.3  717.98     908  786.33   936.8  801.73  1042.4  852.93  1061.6   861.5
#Mann= 3 , 0 , 0
       0     .08       0     533    .045       0     563      .1       0
Bank Sta=533,563
XS Rating Curve= 0 ,0
Exp/Cntr=0.3,0.1

Type RM Length L Ch R = 1 ,5750.4  ,494,494.7,495.4
XS GIS Cut Line= 3
     1872746.312      565143.453     1872374.621       565221.17
     1871752.884      565484.732
#Sta/Elev= 30
       0  824.54    87.6  839.62    97.4  839.41   107.1   835.7   155.8  804.21
   165.5  800.04   194.7  792.43   204.5   788.9   214.2  784.22   311.6   734.1
   428.7  672.21     507  634.13   516.7  631.93   526.5  632.44   536.3     634
   546.1     635   585.2  636.07   614.6   641.9   663.6  647.12   692.9  653.42
   741.8  669.09   751.6  669.78   761.4  671.63   771.2  675.77   790.8  686.74
   869.1  736.88   888.6  747.72   966.9  788.05   986.5   796.5    1055  817.95
#Mann= 3 , 0 , 0
       0      .1       0     507    .045       0   536.3     .06       0
Bank Sta=507,536.3
XS Rating Curve= 0 ,0
Exp/Cntr=0.3,0.1

Type RM Length L Ch R = 1 ,5254.5  ,584.8,563.5,542.2
XS GIS Cut Line= 3
     1872746.312      564748.109     1872161.744      564805.552
     1871509.596      565055.599
#Sta/Elev= 30
       0  739.02    19.6  732.69    39.2  724.38    58.7  713.65   107.7  681.51
   117.5  677.09   127.3  674.83   146.8  675.39   176.2  681.79   264.3  690.97
   323.1   692.4     372  691.37     421  685.44   528.6  649.86     558  642.74
   666.1  638.37   734.9  633.86   754.6  630.65   764.4  629.38   784.1  631.97
   813.6  640.47   882.5  665.37     912  673.56   921.8  677.55     971  702.26
  1059.6  751.69  1118.6  777.37  1148.1  787.34  1226.8  809.01  1285.8  818.56
#Mann= 3 , 0 , 0
       0     .06       0   754.6    .045       0   784.1      .1       0
Bank Sta=754.6,784.1
XS Rating Curve= 0 ,0
Exp/Cntr=0.3,0.1

Type RM Length L Ch R = 1 ,4691    ,413.4,420.4,428.6
XS GIS Cut Line= 3
     1871982.858      563922.526     1871583.934      564636.602
     1871316.993      564930.575
#Sta/Elev= 30
       0   827.6    19.5  820.35    58.4  808.04   126.6  779.69   165.5  759.72
   204.5  741.59   243.4  719.98   262.9  709.96   282.4  700.71   311.6  688.63
   331.1  681.71   350.6  675.79   418.7  658.99   447.9  650.79   525.8  630.64
   535.6  628.82   545.3  628.29   564.8  630.84   584.2  632.06   671.9  634.12
   681.6  634.74   691.4  636.52   798.5  677.51   827.6  686.92   924.5  730.85
   992.3  758.05  1040.7  775.64  1127.9  804.76  1176.3  822.69    1215  835.19
#Mann= 3 , 0 , 0
       0      .1       0   535.6    .045       0   564.8     .06       0
Bank Sta=535.6,564.8
XS Rating Curve= 0 ,0
Exp/Cntr=0.3,0.1

Type RM Length L Ch R = 1 ,4270.3  ,599.3,599.4,598.3
XS GIS Cut Line= 3
     1871768.452      563728.711     1871399.062      564130.669
     1871013.961      564518.429
#Sta/Elev= 30
       0  845.17    29.2  833.14    58.5  822.28     195  778.09   214.5  769.57
     273  742.08   302.2  726.41   350.9  697.96   370.4  687.67   389.9  679.73
   467.9  650.39   497.2   640.2     533  629.14   545.9   626.7   555.7  626.81
     563  628.02     585  631.08     663  634.43   682.5   636.7     702  642.77
   750.8  659.87   760.6  662.61   819.2  676.09   838.7   679.7     868  683.12
   877.7  685.76   965.5  726.27   994.8  738.18  1053.4   760.4  1092.4  779.21
#Mann= 3 , 0 , 0
       0      .1       0     533    .045       0     563     .06       0
Bank Sta=533,563
XS Rating Curve= 0 ,0
Exp/Cntr=0.3,0.1

Type RM Length L Ch R = 1 ,3671    ,512.9,498.5,484.2
XS GIS Cut Line= 3
       1871311.5      563351.641     1870808.396      563894.115
     1870549.959       564166.92
#Sta/Elev= 30
       0  827.16    29.2  819.53    38.9  815.28    68.1  799.92   175.2  739.48
   233.6  710.87   311.5  675.27   360.2  659.02   369.9   656.6   506.2   634.4
     538  626.65   545.2   625.2   554.9  624.86     568  626.49   652.2  639.92
   759.1  659.11     788  666.25   816.9  678.47   836.2   683.1   845.8  687.75
   855.5  695.88   865.1  706.34   874.8   714.3   903.7  734.41   961.5   778.1
   990.4  797.04  1009.6  807.11  1028.9   815.3  1086.7  833.92  1115.6  845.16
#Mann= 3 , 0 , 0
       0      .1       0     538    .045       0     568     .08       0
Bank Sta=538,568
XS Rating Curve= 0 ,0
Exp/Cntr=0.3,0.1

Type RM Length L Ch R = 1 ,3172.3  ,531.7,539.1,546.5
XS GIS Cut Line= 4
     1870911.512       562876.14     1870563.475      563362.717
     1870485.758      563639.795     1870255.985      563883.084
#Sta/Elev= 30
       0  799.59    29.4  790.42      49  780.78    68.6  772.94   107.9  763.36
   137.3  754.59   176.5   741.4   215.8  726.08   274.6  707.79     304  696.43
   323.6  690.31   372.7  680.32   431.5   672.2     510  653.65   665.4  633.14
   690.6  625.97   703.8  623.73   720.6  625.83   742.1  631.94   790.1  640.97
   915.5  659.37   974.6  679.23    1014  689.33  1033.6  701.18  1102.5  749.58
  1141.9  774.73  1161.6  785.81  1181.3  799.17    1201  807.71  1220.6  812.42
#Mann= 3 , 0 , 0
       0     .08       0   690.6    .045       0   720.6      .1       0
Bank Sta=690.6,720.6
XS Rating Curve= 0 ,0
Exp/Cntr=0.3,0.1

Type RM Length L Ch R = 1 ,2633.1  ,530.6,532.9,535.2
XS GIS Cut Line= 3
     1870342.094      562784.112     1870002.504      563351.785
     1869797.229      563698.977
#Sta/Elev= 30
       0  830.28    58.4  803.52    87.6  787.54   116.7  766.87   155.6  733.47
   175.1     720   194.6  708.68     214   699.8   272.4  678.73   379.4  630.92
   389.1  627.99   398.8  626.92   486.4  626.78   505.5  624.43   525.3  622.08
   535.5  624.59   554.5   631.1   593.4  632.94   661.5  640.98   779.5  661.55
   799.2  666.26   828.7  677.45   848.4   682.2   858.2  685.48   868.1  690.95
   897.6  710.18   966.5  757.77  1005.8  782.38  1015.6  786.91  1064.8  801.73
#Mann= 3 , 0 , 0
       0     .08       0   505.5    .045       0   535.5     .08       0
Bank Sta=505.5,535.5
XS Rating Curve= 0 ,0
Exp/Cntr=0.3,0.1
